--- NFSBPOTMC_T1.prj (project) ---

Proj Title=NFSBPOTMC_T1
Current Plan=p01
Default Exp/Contr=0,0
English Units
Geom File=g01
Flow File=f01
Plan File=p01
BEGIN DESCRIPTION:
Stream Name: North Fork South Branch Potomac River Tributary 1
Flood Zone: Approximate
Pendleton County, West Virginia
HEC-RAS Version: 5.0.7
Hydrology Method:
Regression equation
END DESCRIPTION:
DSS Export Rating Curves= 0
DSS Export Rating Curve Sorted= 0
DSS Export Volume Flow Curves= 0
DXF OffsetX= 0
DXF OffsetY= 0
DXF ScaleX= 0
DXF ScaleY= 0

--- NFSBPOTMC_T1.p01 (plan) ---

Plan Title=Floodplain
Program Version=5.07
Short Identifier=Floodplain
Geom File=g01
Flow File=f01
Subcritical Flow
K Sum by GR= 0
Std Step Tol= 0.01
Critical Tol= 0.01
Num of Std Step Trials= 20
Max Error Tol= 0.3
Flow Tol Ratio= 0.001
Split Flow NTrial= 30
Split Flow Tol= 0.02
Split Flow Ratio= 0.02
Log Output Level= 0
Friction Slope Method= 1
Unsteady Friction Slope Method= 2
Unsteady Bridges Friction Slope Method= 1
Parabolic Critical Depth
Global Vel Dist= 0 , 0 , 0
Global Log Level= 0
CheckData=False
Encroach Param=-1 ,0,0, 0
Mapping Interval=1HOUR
Computation Time Step Use Courant=        0
Computation Time Step Use Time Series=    0
Computation Time Step Count To Double=0
Computation Time Step Max Doubling=0
Computation Time Step Max Halving=0
Computation Time Step Residence Courant=0
Run HTab= 0
Run UNet= 0
Run Sediment= 0
Run PostProcess= 0
Run WQNet= 0
Run RASMapper= 0
UNET Theta= 0
UNET Theta Warmup= 0
UNET ZTol= 0
UNET ZSATol= 0
UNET MxIter= 0
UNET Max Iter WO Improvement= 0
UNET MaxInSteps= 0
UNET DtIC= 0
UNET DtMin= 0
UNET MaxCRTS= 0
UNET WFStab= 0
UNET SFStab= 0
UNET WFX= 1
UNET SFX= 1
UNET 1D Methodology=Finite Difference
UNET DSS MLevel= 1
UNET Pardiso=0
UNET DZMax Abort= 0
UNET Use Existing IB Tables= 0
UNET Froude Reduction=False
UNET Froude Limit= 0
UNET Froude Power= 0
UNET D1 Cores= 0
UNET D2 Coriolis=0
UNET D2 Cores= 0
UNET D2 Theta= 1
UNET D2 Theta Warmup= 1
UNET D2 Z Tol= 0.01
UNET D2 Volume Tol= 0.01
UNET D2 Max Iterations= 20
UNET D2 Equation= 0
UNET D2 RampUpFraction=0.1
UNET D2 TimeSlices= 1
UNET D2 BCVolumeCheck=0
UNET D1D2 MaxIter= 0
UNET D1D2 ZTol=0.01
UNET D1D2 QTol=0.1
UNET D1D2 MinQTol=1
Write IC File= 0
Write IC File at Fixed DateTime=0
Write IC File at Sim End=0
Echo Input=False
Echo Parameters=False
Echo Output=False
Write Detailed= 0
HDF Write Warmup=0
HDF Write Time Slices=0
HDF Flush=0
HDF Face Node Velocities=0
HDF Compression= 1
HDF Chunk Size= 1
HDF Spatial Parts= 1
HDF Use Max Rows=0
HDF Fixed Rows= 1
Calibration Method= 0
Calibration Iterations= 20
Calibration Max Change=0.05
Calibration Tolerance=0.2
Calibration Maximum=1.5
Calibration Minimum=0.5
Calibration Optimization Method= 1
WQ AD Non Conservative
WQ ULTIMATE=-1
WQ Max Comp Step=1HOUR
WQ Output Interval=15MIN
WQ Output Selected Increments= 0
WQ Output face flow=0
WQ Output face velocity=0
WQ Output face area=0
WQ Output face dispersion=0
WQ Output cell volume=0
WQ Output cell surface area=0
WQ Output cell continuity=0
WQ Output cumulative cell continuity=0
WQ Output face conc=0
WQ Output face dconc_dx=0
WQ Output face courant=0
WQ Output face peclet=0
WQ Output face adv mass=0
WQ Output face disp mass=0
WQ Output cell mass=0
WQ Output cell source sink temp=0
WQ Output nsm pathways=0
WQ Output nsm derived pathways=0
WQ Output MaxMinRange=-1
WQ Daily Max Min Mean=-1
WQ Daily Range=0
WQ Daily Time=0
WQ Create Restart=0
WQ Fixed Restart=0
WQ System Summary=0
WQ Write To DSS=0
WQ Use Fixed Temperature=0
Sorting and Armoring Iterations= 10
XS Update Threshold= 0.02
Bed Roughness Predictor= 0
Hydraulics Update Threshold= 0.02
Energy Slope Method= 1
Volume Change Method= 1
Sediment Retention Method= 0
XS Weighting Method= 0
Number of US Weighted Cross Sections= 1
Number of DS Weighted Cross Sections= 1
Upstream XS Weight=0
Main XS Weight=1
Downstream XS Weight=0
Number of DS XS's Weighted with US Boundary= 1
Upstream Boundary Weight= 1
Weight of XSs Associated with US Boundary= 0
Number of US XS's Weighted with DS Boundary= 1
Downstream Boundary Weight= 0.5
Weight of XSs Associated with DS Boundary= 0.5
Percentile Method= 0
Sediment Output Level= 3
Mass or Volume Output= 0
Output Increment Type= 1
Profile and TS Output Increment= 1
XS Output Flag= 0
XS Output Increment= 10
Write Gradation File= 0
Read Gradation Hotstart= 0
Write HDF5 File= 1
Write Binary Output= 1
Write DSS Sediment File= 0
SV Curve= 0
Specific Gage Flag= 0

--- NFSBPOTMC_T1.f01 (steady flow) ---

Flow Title=Flows
Program Version=5.07
Number of Profiles= 6
Profile Names=P100yr,P10yr,P25yr,P50yr,P500yr,P101yr
River Rch & RM=NFSBPOTMC_T1,Main            ,10594
     327     154     217     271     477     398
River Rch & RM=NFSBPOTMC_T1,Main            ,9882
     632     295     418     522     928     770
River Rch & RM=NFSBPOTMC_T1,Main            ,6793
     806     375     531     665    1186     981
River Rch & RM=NFSBPOTMC_T1,Main            ,4335
    1455     671     955    1198    2154    1771
Boundary for River Rch & Prof#=NFSBPOTMC_T1,Main            , 1
Up Type= 0
Dn Type= 3
Dn Slope=0.01698
Boundary for River Rch & Prof#=NFSBPOTMC_T1,Main            , 2
Up Type= 0
Dn Type= 3
Dn Slope=0.01698
Boundary for River Rch & Prof#=NFSBPOTMC_T1,Main            , 3
Up Type= 0
Dn Type= 3
Dn Slope=0.01698
Boundary for River Rch & Prof#=NFSBPOTMC_T1,Main            , 4
Up Type= 0
Dn Type= 3
Dn Slope=0.01698
Boundary for River Rch & Prof#=NFSBPOTMC_T1,Main            , 5
Up Type= 0
Dn Type= 3
Dn Slope=0.01698
Boundary for River Rch & Prof#=NFSBPOTMC_T1,Main            , 6
Up Type= 0
Dn Type= 3
Dn Slope=0.01698
DSS Import GetInterval= 0
DSS Import GetPeak= 0
DSS Import FillOption= 0

--- NFSBPOTMC_T1.g01 (geometry) ---

Geom Title=Geometry
Program Version=5.07

River Reach=NFSBPOTMC_T1    ,Main
Reach XY= 30
2433312.42162573666157.2368801532433123.19168928 665970.92885381
2433001.95997635665670.9796505872432779.77997448 665535.01043433
2432861.90448223665318.5020090642432787.00436954665019.163040876
2432628.56308536664891.392299026 2432542.6105013664599.376806915
2432611.77342071664353.5990832452432558.69905183664109.340057328
2432395.72792108664063.1095067412431871.04885237663365.760507748
2431621.44108388663228.1469378172431539.42812449662905.678750739
2430764.39752238662741.8027661892430472.24817225662284.002172589
2430180.61555347662109.976602018 2429845.3859089662064.630892187
2429570.59479186662362.2999162522429312.28330061662445.809263662
2429115.09767139662775.9831439852428990.88991448662833.878041312
 2428741.0180389662831.5443845842428536.07553548662613.845344886
2428221.70313264662567.056396499 2427877.2504095662393.990469679
2427460.52289656662342.1191823332427062.81667092662146.210453391
 2426672.0625312662157.1326756632426189.64152244662425.447472081

Type RM Length L Ch R = 1 ,10594   ,204.2,204.5,205
XS GIS Cut Line= 3
     2433618.402       665885.68     2433305.969      666149.598
2433122.55196846666323.562017641
#Sta/Elev= 30
       0 2005.06    20.5 2014.07    60.2 2038.62    76.3 2040.87    82.5 2043.57
    88.7 2047.75   101.1 2060.42   119.8 2067.79   142.5 2068.48   182.8 2059.61
   198.5 2049.36     209 2045.51   236.2 2044.15   250.9 2035.81   301.5  2017.3
     327 2004.39   361.4 1998.81   375.3 1990.35   392.4 1989.73   397.5 1987.53
   402.7 1981.77     408 1980.02   416.51981.933   437.6 1990.31     469  1993.4
   480.1 1996.47   512.7 2011.63   545.7 2033.09   578.8 2051.45   661.8    2087
#Mann= 5 ,-1 , 0
       0      .1       0  316.13     .06       0   402.7    .045       0
   416.5     .06       0  478.07      .1       0
Bank Sta=402.7,416.5
XS Rating Curve= 0 ,0
Exp/Cntr=0.3,0.1

Type RM Length L Ch R = 1 ,10389   ,52.5,57.5,61.5
XS GIS Cut Line= 3
2433408.02426876665783.9231326922433194.86110034665981.347237637
2433038.94589188666106.866712458
#Sta/Elev= 30
       0 2007.42     5.8 2006.77    10.3 2005.24    34.1 1983.21    39.8  1981.1
    45.6 1981.67    48.3 1982.75    86.8 2001.33    92.7 2003.94    98.6 2005.17
   215.3 1996.19   225.3 1995.42   241.6 1995.76   252.5 1992.32   271.9 1983.92
   280.4 1981.76   291.7 1977.37     301 1975.66   325.9 1975.62   332.9 1972.88
   337.2 1971.23   340.1 1971.15   347.2 1973.13   357.4 1981.49   362.8 1984.81
   382.3 1994.43   393.4 1997.79   401.4  2002.9   424.2 2014.48   490.7 2050.79
#Mann= 4 ,-1 , 0
       0      .1       0   215.3     .06       0   332.9    .045       0
   347.2      .1       0
Bank Sta=332.9,347.2
XS Rating Curve= 0 ,0
Exp/Cntr=0.5,0.3

Type RM Length L Ch R = 1 ,10332   ,59.4,58.8,58.9
XS GIS Cut Line= 4
2433373.62799466665741.6375818552433180.02255559665968.435481446
2433087.53382109 665965.201609612433026.09025621666095.203257411
#Sta/Elev= 30
       0 2005.56      20 2004.41    38.5    2001      49  1996.7    64.8 1983.67
    75.3 1980.06    91.1 1980.97     103 1986.91   112.1 1989.59   159.4 1998.01
   222.5 1995.89   248.8 1996.66   258.3 1995.24   269.4 1990.62   280.4 1985.02
   296.2  1974.8   303.5 1973.79   339.4 1973.84   348.51970.559   355.5 1968.63
   361.21970.456   367.5 1975.35   371.5 1976.97   392.6 1977.66   416.6 1980.41
     428 1983.82   439.4 1990.13   476.8 2016.55   494.7    2028   534.5 2050.24
#Mann= 5 ,-1 , 0
       0      .1       0  213.86     .06       0   348.5    .045       0
   361.2     .06       0  447.64      .1       0
#XS Ineff= 2 , 0
          339.43  1973.7   365.3          1973.3
Permanent Ineff=
       F       F
Bank Sta=348.5,361.2
XS Rating Curve= 0 ,0
Exp/Cntr=0.5,0.3

Type RM Length L Ch R = 1 ,10273   ,48.8,38.1,31.8
XS GIS Cut Line= 4
2433350.89925816665717.4764078052433174.59796417 665909.52099354
2433091.41446729665906.3451421982433008.52076378666092.520422588
#Sta/Elev= 30
       0 2004.25    18.2 2003.14    60.6 1997.81    67.1 1995.62    80.4 1986.43
    91.7 1982.88   100.8 1977.46   110.5 1974.96   121.4 1975.14   126.8 1976.38
   148.1 1983.31   164.8 1989.95   186.5  1994.2   213.7 1994.67   254.6 1993.37
   260.5  1992.1   264.6  1989.7   284.6 1972.61   295.3 1968.71   304.6 1967.22
   316.91968.892   324.6 1971.74   355.4 1971.04   375.2    1972   392.7 1977.14
   423.4 1979.17   432.1 1981.83   441.8 1987.36     489 2021.66   547.7 2055.62
#Mann= 5 ,-1 , 0
       0      .1       0  289.03     .06       0   295.3    .045       0
   316.9     .06       0  426.98      .1       0
Bank Sta=295.3,316.9
XS Rating Curve= 0 ,0
Exp/Cntr=0.5,0.3

Type RM Length L Ch R = 1 ,10235   ,36.6,32.3,30.6
XS GIS Cut Line= 3
2433312.58057908665669.8711695122433077.15470943665907.237362263
 2432993.0740417666079.926118297
#Sta/Elev= 30
       0 2003.89      14  2003.3    97.2 1995.91   125.4 1991.62   142.3 1987.74
   159.2 1982.74   180.2 1972.85   198.6 1968.06   207.1 1967.69   249.3 1971.44
   263.9 1971.62   269.6 1970.28   274.81966.968   280.9 1965.69   294.71967.228
     300  1969.6   303.7 1970.48   339.8 1970.28   356.2 1971.35   371.8 1974.32
   380.7 1977.11   400.7 1978.06   407.7 1979.36   413.7  1981.3   422.1 1985.67
   432.4 1992.45   467.7 2019.73   485.2 2031.81   511.9 2048.32   526.4  2056.6
#Mann= 5 ,-1 , 0
       0      .1       0  250.17     .06       0   274.8    .045       0
   294.7     .06       0  388.59      .1       0
#XS Ineff= 2 , 0
          258.22 1974.77
Permanent Ineff=
       F       F
Bank Sta=274.8,294.7
XS Rating Curve= 0 ,0
Exp/Cntr=0.5,0.3

Type RM Length L Ch R = 1 ,10203   ,53.5,55.1,54.6
XS GIS Cut Line= 3
2433149.29465778665549.2894356182433117.06010019665798.233443327
2432980.64151109666077.652019322
#Sta/Elev= 30
       0 2003.79    33.9 1999.64      46 1996.01    58.1 1988.77    78.2 1968.43
    82.3 1966.14    86.3 1965.51    94.4 1965.24    98.4 1967.07   107.3 1973.93
   118.6 1978.53   142.8 1977.65   158.9 1984.28     163 1984.92   199.3 1975.41
   219.4 1971.41   243.6 1972.33   290.9 1964.61   296.3 1963.42   304.1 1963.39
     311 1964.25     323 1969.43   381.9 1970.49   403.1 1976.22   434.3 1978.18
   441.7 1980.19   456.9 1988.06     501 2021.05   527.7 2039.97     562 2061.15
#Mann= 6 ,-1 , 0
       0      .1       0  211.73    .055       0   281.9     .06       0
   290.9    .045       0     311     .06       0  403.74      .1       0
#XS Ineff= 2 , 0
          280.57  1967.6  316.45          1968.2
Permanent Ineff=
       F       F
Bank Sta=290.9,311
XS Rating Curve= 0 ,0
Exp/Cntr=0.5,0.3

Type RM Length L Ch R = 1 ,10148   ,44.1,48.8,54
XS GIS Cut Line= 3
 2433105.0519496665541.2927028482433070.88775172665772.805067825
2432946.74164471666045.428039487
#Sta/Elev= 30
       0 1998.45    46.1 1994.16    75.1 1988.86    82.5 1985.42    86.5 1982.21
   102.7 1964.28   106.7 1961.64   110.8 1960.22   118.9 1959.56     127  1960.8
   146.2 1965.69   159.3 1970.12   179.6 1970.32   240.7 1967.51   247.8 1965.97
   263.71958.712   271.5 1957.09   275.9 1957.61   279.1 1959.01   289.1 1965.53
   297.8 1968.17   346.2 1969.39   368.2 1978.98     377 1981.46   398.8 1985.49
   420.9 1992.84   438.5 2002.18   486.8 2034.91     522  2055.4   533.6  2060.7
#Mann= 6 ,-1 , 0
       0      .1       0  192.16    .055       0   263.7    .045       0
   279.1    .055       0  302.89     .06       0  318.01      .1       0
#XS Ineff= 2 , 0
          171.25 1979.29
Permanent Ineff=
       F       F
Bank Sta=263.7,279.1
XS Rating Curve= 0 ,0
Exp/Cntr=0.5,0.3

Type RM Length L Ch R = 1 ,10099   ,217.9,216.3,210.6
XS GIS Cut Line= 3
 2433081.4417007665505.0835259192433054.62284286665751.862730106
2432796.95778331665897.982310724
#Sta/Elev= 30
       0 1996.84    46.1  1994.3    74.2 1991.54    94.8 1987.68   126.5 1983.67
   134.6 1980.57   142.6 1975.46   154.7 1964.13   158.7 1961.21   166.8 1958.73
   186.9 1959.54   197.6 1962.11   215.1 1964.69   243.2 1966.24   248.2 1965.93
   261.9 1961.87   272.71956.871   280.3 1955.57   291.4 1956.73   306.1 1959.43
   326.3 1970.85   332.5  1971.8   353.1 1971.88   367.7 1980.12   379.5 1982.64
   392.2  1987.1   420.6 2001.15   491.8  2040.9   533.2  2061.2   544.4 2065.44
#Mann= 5 ,-1 , 0
       0      .1       0  230.84    .055       0   272.7    .045       0
   291.4     .06       0   390.3      .1       0
#XS Ineff= 2 , 0
          231.53  1971.2
Permanent Ineff=
       F       F
Bank Sta=272.7,291.4
XS Rating Curve= 0 ,0
Exp/Cntr=0.3,0.1

Type RM Length L Ch R = 1 ,9882    ,160.3,166,171.5
XS GIS Cut Line= 3
2433283.25120809665392.9621470582432974.12772026665531.702610099
2432712.46807505665860.298443618
#Sta/Elev= 30
       0  2020.3   149.6 2006.97   202.2 2000.43   285.5 1988.14   307.5    1984
   343.5 1974.13   376.4 1968.74   403.3 1959.82     409 1958.78   420.4 1958.39
   426.1  1957.6   429.8 1956.33   445.2 1948.37   455.4  1941.9   460.5 1940.72
   470.7  1940.5   475.9 1940.61     481 1941.71   491.2 1947.05   511.6 1963.29
   528.5  1973.8   531.4 1975.07   534.2 1975.54   549.7 1975.38   554.2 1976.53
   562.7 1982.29   588.3 1992.34   653.8 2023.47   703.9 2049.36   758.9 2079.13
#Mann= 4 ,-1 , 0
       0      .1       0   455.4    .045       0     481     .06       0
  593.25      .1       0
Bank Sta=455.4,481
XS Rating Curve= 0 ,0
Exp/Cntr(USF)=0,0
Exp/Cntr=0.3,0.1

Type RM Length L Ch R = 1 ,9716    ,321.6,322.5,324.5
XS GIS Cut Line= 3
2433113.47407622665382.6119375732432965.79796772665470.875007615
2432437.15545442665630.779308268
#Sta/Elev= 30
       0 2002.42    31.1 1999.41    82.4 1990.97   152.3 1978.35   183.6 1971.33
   212.8 1967.39   251.5 1954.84   283.9 1948.71   292.2 1947.97   321.5 1949.47
   329.9 1948.81   338.4 1946.21   354.2 1936.78   359.1 1935.17   367.5 1933.46
   375.8 1934.02   379.3 1935.71   384.2 1940.44   392.5 1951.78   396.7  1956.2
   400.9 1958.08   417.6  1958.6   421.8 1959.88   438.5 1974.76   476.1    1998
   534.6 2036.33     543 2040.91   630.1 2100.43   718.5 2167.36   724.3 2172.52
#Mann= 4 ,-1 , 0
       0      .1       0   359.1    .045       0   379.3     .06       0
  463.74      .1       0
Bank Sta=359.1,379.3
XS Rating Curve= 0 ,0
Exp/Cntr=0.3,0.1

Type RM Length L Ch R = 1 ,9394    ,355.6,344.7,335.5
XS GIS Cut Line= 3
2433238.56662084665171.991104201     2432838.937       665232.49
2432401.60481881665303.619825761
#Sta/Elev= 30
       0 2023.15   161.6 1992.15   181.9 1987.61   198.1  1979.9   222.3 1977.84
   254.7 1967.73   297.5 1958.24   323.5 1955.26   339.6 1950.18   355.8  1949.1
   376.1 1933.61   388.2 1921.47     392 1918.89   408.4 1917.46   412.5 1918.83
   420.6 1923.98   436.8 1927.48   457.1 1934.12   465.2 1935.26   578.6 1934.65
   582.7 1937.28   590.8 1946.59   598.9 1953.96   612.1 1961.99     626 1974.84
     684 2023.66     748 2071.12     761 2077.62   775.9  2090.9   847.3 2144.62
#Mann= 6 ,-1 , 0
       0     .05       0  109.64      .1       0     392    .045       0
   412.5    .055       0  506.92     .06       0  606.23      .1       0
Bank Sta=392,412.5
XS Rating Curve= 0 ,0
Exp/Cntr=0.3,0.1

Type RM Length L Ch R = 1 ,9049    ,96.1,105.3,112.5
XS GIS Cut Line= 4
2433087.91279464664839.7276804992432707.86887546664892.543451744
2432690.64634136665014.2493593952432319.78777371665141.696111747
#Sta/Elev= 30
       0 2022.11    41.6 2005.58    98.1 1980.48   146.6 1961.67   158.7 1955.66
   170.8 1953.83   235.4 1925.48   243.5 1926.73   332.3 1925.88   364.6  1922.6
   372.6  1919.9   386.1 1911.72   402.2 1910.48   417.61902.988   426.5  1901.6
   432.2 1902.16   450.7 1903.81   499.2 1915.21     515  1916.9   550.5 1924.33
   578.4 1926.08   627.9 1955.34   654.5  1974.7   667.2 1984.63   680.2 1991.97
   701.1  2009.3   713.8 2016.88   857.6 2124.58   870.3 2130.72   898.8 2151.09
#Mann= 6 ,-1 , 0
       0     .05       0   146.6      .1       0   417.6    .045       0
   432.2    .055       0   550.5     .06       0   654.5      .1       0
Bank Sta=417.6,432.2
XS Rating Curve= 0 ,0
Exp/Cntr(USF)=0,0
Exp/Cntr=0.3,0.1

Type RM Length L Ch R = 1 ,8944    ,259.1,260.6,260.6
XS GIS Cut Line= 3
2433069.24645442664762.961881344     2432622.255      664875.035
     2432231.008      664966.261
#Sta/Elev= 30
       0 2030.43    43.8  2011.7   113.9  1977.4   159.3 1957.23   167.5 1950.98
   179.9 1948.38   203.1 1935.28   225.3 1926.25   373.7 1923.53   381.2 1921.15
   394.3 1911.72   410.8 1907.95   427.3 1895.97   433.9 1894.61   453.6 1896.58
   460.4 1895.06     467 1896.62   480.3  1910.7     485 1913.42   516.9  1912.9
     526 1916.92   587.7 1966.76   612.3 1988.36   628.7 1997.16   650.1 2017.02
   690.1 2049.92   700.1 2055.91   713.4 2067.09   751.9 2093.65   862.6 2164.51
#Mann= 7 ,-1 , 0
       0      .1       0  107.66     .05       0  307.01    .055       0
  406.69     .06       0   453.6    .045       0     467     .06       0
   506.3      .1       0
Bank Sta=453.6,467
XS Rating Curve= 0 ,0
Exp/Cntr=0.3,0.1

Type RM Length L Ch R = 1 ,8683    ,337,338.8,338.4
XS GIS Cut Line= 2
     2432987.542      664559.107     2432155.926      664712.579
#Sta/Elev= 30
       0 2012.61    94.4  1959.6   106.6 1954.72   155.4 1929.18   171.6 1927.52
   192.8  1921.5   228.6 1916.95   269.3 1913.25   301.8 1913.48   346.6 1909.06
     375 1901.92   411.6 1896.47   427.9 1889.19   433.2 1883.47     440 1881.57
   452.3 1882.99   457.2 1884.24   464.1 1888.61   480.1 1905.59   484.8 1908.81
   505.2 1910.55   522.4 1930.18   589.9 1971.95   642.6 2007.32   659.8 2014.55
   679.6 2027.98   785.8    2093   830.6 2124.18   838.7 2126.35   845.7 2131.38
#Mann= 7 ,-1 , 0
       0      .1       0   59.26     .05       0  257.94    .055       0
  357.28     .06       0   433.2    .045       0   452.3     .06       0
  555.96      .1       0
Bank Sta=433.2,452.3
XS Rating Curve= 0 ,0
Exp/Cntr=0.3,0.1

Type RM Length L Ch R = 1 ,8345    ,259.6,251.3,230.8
XS GIS Cut Line= 2
     2433006.343      664299.2582432146.71949445664356.730527731
#Sta/Elev= 30
       0 2028.81    47.7 2017.83    75.8 2008.73   139.9 1994.39   187.2 1979.19
   197.6 1974.38   236.1 1951.55   288.2 1923.63   330.8 1907.79   340.4  1902.8
   360.4 1900.73   372.4 1892.49   386.3 1875.22   390.1 1871.75   392.5 1870.37
   400.5 1869.86   410.61871.676   420.5 1877.07   436.6 1879.18   456.6 1885.71
   528.8 1887.61   584.9  1884.8     613 1886.77     645 1904.35   665.1  1911.9
   681.1  1916.2   741.2 1947.31   777.3 1964.13   853.5 1987.23   861.5 1992.38
#Mann= 7 ,-1 , 0
       0      .1       0  319.43     .05       0   390.1    .045       0
   410.6     .05       0  419.19      .1       0  518.95     .06       0
   618.7      .1       0
Bank Sta=390.1,410.6
XS Rating Curve= 0 ,0
Exp/Cntr=0.3,0.1

Type RM Length L Ch R = 1 ,8093    ,84.4,82.2,76.8
XS GIS Cut Line= 4
2432811.81772849663776.1262896922432569.53640631 664005.89298985
2432488.42252251664245.0230299812432233.52308197664297.615787154
#Sta/Elev= 30
       0 1899.28      31 1902.09   104.6 1897.71   195.8 1896.77   224.9 1898.91
   248.2 1895.92   277.1  1896.8   299.2 1891.36   315.7 1890.89   333.9 1883.63
   364.5 1878.01   377.9 1873.58   406.8 1874.69     411 1871.83   418.21862.842
   427.9  1861.2   444.41862.679   470.1 1869.49   516.7 1871.77   541.9 1877.35
   579.9 1881.25     629 1877.82   665.7 1879.01   686.2 1889.08   714.7 1908.88
     727  1915.4   768.9 1927.76   792.3 1936.87   804.6 1939.28   846.7 1952.86
#Mann= 6 ,-1 , 0
       0      .1       0   38.79     .05       0  210.34      .1       0
   418.2    .045       0   444.4      .1       0  620.24     .06       0
Bank Sta=418.2,444.4
XS Rating Curve= 0 ,0
Exp/Cntr=0.5,0.3

Type RM Length L Ch R = 1 ,8011    ,48.6,48.8,50.2
XS GIS Cut Line= 4
      2432715.53      663734.824 2432462.1242834664014.202938055
2432457.68138644664200.988429657 2432189.3740136664261.047379229
#Sta/Elev= 30
       0 1887.76    17.6 1892.46    37.4 1894.58   151.3 1885.99   215.8 1886.83
   257.2 1882.36   286.3 1871.12   304.8 1867.95   361.9 1864.91   377.2 1862.32
   397.9 1865.62   413.9 1865.52     432 1859.46   441.9 1857.05   456.31859.554
   489.9 1867.78   521.9 1868.62   545.9 1875.86     564 1878.63   591.6 1874.07
   612.1 1874.49   632.6 1878.33   648.5 1886.08   681.9 1910.98   694.1 1917.52
   735.1 1928.79   779.1 1935.64   796.6 1940.38   817.1 1947.31     839 1957.33
#Mann= 6 ,-1 , 0
       0      .1       0   28.11     .05       0  278.62      .1       0
     432    .045       0   456.3      .1       0  514.97     .06       0
#XS Ineff= 2 ,-1
       0  423.98 1862.42  466.13     649  1863.4
Permanent Ineff=
       F       F
Bank Sta=432,456.3
XS Rating Curve= 0 ,0
Exp/Cntr=0.5,0.3

Type RM Length L Ch R = 1 ,7962    ,74.8,83,91.5
XS GIS Cut Line= 4
        2432689.      663705.755  2432415.050517 664011.25965668
2432407.83089551664166.0930860042432138.87397292664234.024437349
#Sta/Elev= 30
       0 1878.22      23 1883.64    33.8  1887.6    55.3 1890.66   114.4  1888.4
   189.1 1880.47   237.9 1882.62   264.8 1879.92     285 1868.31   305.5 1862.42
   384.8 1859.11     442 1859.32     454 1856.42   463.41851.572     470 1850.33
   479.91852.063     502 1869.65   526.1 1873.02   565.3 1872.51   591.2 1876.19
   603.6 1881.71   636.6 1904.78   649.2 1911.41   669.6 1917.27   686.1 1920.11
   727.4 1924.09   743.9 1930.69   752.1 1932.29   809.9 1965.16   842.7 1985.62
#Mann= 7 ,-1 , 0
       0      .1       0     .57      .1       0   20.39     .05       0
  328.47      .1       0  383.46     .06       0   463.4    .045       0
   479.9     .06       0
Bank Sta=463.4,479.9
XS Rating Curve= 0 ,0
Exp/Cntr=0.5,0.3

Type RM Length L Ch R = 1 ,7879    ,446.6,445.2,440.7
XS GIS Cut Line= 3
2432674.53803474  663678.09886052432400.63886745663989.668700157
2432049.56458525664168.485738642
#Sta/Elev= 30
       0 1884.19    27.7 1875.72    34.4 1876.77      49 1883.67    85.4 1888.11
   155.5 1885.83   224.7 1877.38     278 1877.56     315 1860.52     383 1860.35
   393.5 1857.56   425.9 1856.66     438 1848.47   443.9 1846.72   457.4 1848.56
   470.8 1856.02   494.5 1864.68   515.7 1869.06     548 1887.34     592 1898.04
   614.5 1907.84   637.9 1920.57   655.1 1932.08   668.4  1936.9   681.8 1947.23
   744.7 1986.85   753.6  1994.2   767.1 1998.55     777 2006.94   808.8 2026.81
#Mann= 7 ,-1 , 0
       0      .1       0   66.26     .05       0  370.69      .1       0
  373.79     .06       0     438    .045       0   457.4     .06       0
  485.86      .1       0
Bank Sta=438,457.4
XS Rating Curve= 0 ,0
Exp/Cntr=0.3,0.1

Type RM Length L Ch R = 1 ,7434    ,330.9,330.5,330.6
XS GIS Cut Line= 2
     2432400.015      663410.9942431818.36743727663951.856423964
#Sta/Elev= 30
       0 1894.77    26.3 1878.91    60.3 1848.22    67.3 1844.85    74.4 1845.09
   105.5 1854.74   133.8 1858.32   187.6 1858.91   225.7 1856.47   242.1 1845.77
   326.3  1847.3   345.8 1845.92   354.6 1843.05   408.4 1842.94     431 1829.52
   438.7 1826.58     448 1823.93   453.7 1826.05   467.8 1842.09   476.9 1858.78
   487.6 1872.88   510.9 1892.99   549.9 1914.06   558.9 1917.02   600.8 1947.37
   651.7 1978.77   694.2 2000.79   705.6 2003.57   739.5 2022.63   794.3 2049.73
#Mann= 6 ,-1 , 0
       0      .1       0   72.49     .05       0  273.82     .06       0
  430.66      .1       0   438.7    .045       0   453.7      .1       0
Bank Sta=438.7,453.7
XS Rating Curve= 0 ,0
Exp/Cntr=0.3,0.1

Type RM Length L Ch R = 1 ,7104    ,312.8,311,310.9
XS GIS Cut Line= 2
     2432234.514      663164.1562431606.14680492663695.328435597
#Sta/Elev= 30
       0 1875.67    30.2 1866.94      73 1851.79      91  1847.3   114.9 1844.16
   140.5 1842.78   235.4 1840.26   289.3 1837.45     314 1833.37   324.4 1828.53
   332.6  1822.8   345.2 1819.42   370.8 1818.33     382 1820.67     385 1820.12
   399.1 1811.42   413.2 1809.64   419.71811.283   462.7 1852.92     507 1881.92
   528.7 1894.26   570.6 1912.89   581.1 1915.08   617.6 1930.86   708.5 1963.89
   738.2 1976.07   751.1 1982.57   759.6 1983.62   769.6 1990.37   822.8 2017.34
#Mann= 5 ,-1 , 0
       0     .05       0  273.44    .055       0  389.31      .1       0
   399.1    .045       0   419.7      .1       0
Bank Sta=399.1,419.7
XS Rating Curve= 0 ,0
Exp/Cntr=0.3,0.1

Type RM Length L Ch R = 1 ,6793    ,104.5,110.9,114.9
XS GIS Cut Line= 2
2432011.36688347662949.2241411772431394.83713993663518.263322144
#Sta/Elev= 30
       0 1845.24    12.9 1839.97    46.9 1835.71    67.3 1830.45    80.9 1831.12
   202.3 1827.34     296 1822.45   332.9 1822.71   381.9 1819.32   395.1 1815.62
   414.5 1806.47   452.6 1806.18   460.31802.815   468.7 1800.24   474.3 1801.05
   477.2 1803.23   486.1 1813.27   499.8 1838.21   512.5 1855.75   521.4  1865.3
   533.2 1874.09   615.8 1903.57   637.7 1913.83   726.3 1959.51   739.7 1964.66
   757.4 1975.16   765.9 1976.84     775 1983.73   828.1 2015.02     839 2018.31
#Mann= 5 ,-1 , 0
       0     .05       0  326.07    .055       0   460.3    .045       0
   477.2    .055       0  501.07      .1       0
Bank Sta=460.3,477.2
XS Rating Curve= 0 ,0
Exp/Cntr=0.5,0.3

Type RM Length L Ch R = 1 ,6682    ,95.6,96.1,95.5
XS GIS Cut Line= 4
2432002.95894312662943.031302389 2431638.1518653663174.802907166
2431445.98903281663212.2370555442431401.95371418663328.565859956
#Sta/Elev= 30
       0 1845.72    11.6 1840.38      58 1832.81    71.3 1828.76      95 1827.53
   126.5 1828.37   199.3 1825.95   235.1 1824.13   265.6 1821.11   374.6 1817.33
   384.1 1815.41   402.9 1813.99     422 1804.18   447.9 1802.89   455.61798.219
   468.3 1796.02   472.4 1796.43   474.91798.722   484.6 1807.75     505 1813.85
   517.2 1819.85   529.4 1828.42   545.7 1835.98   557.9 1838.24   570.2 1843.15
   594.6 1849.44     616 1854.13     628  1855.2   638.8 1858.69   752.4 1915.82
#Mann= 5 ,-1 , 0
       0     .05       0  369.05     .06       0   455.6    .045       0
   474.9     .05       0   572.9      .1       0
#XS Ineff= 2 , 0
          448.68 1802.29  479.47          1801.7
Permanent Ineff=
       F       F
Bank Sta=455.6,474.9
XS Rating Curve= 0 ,0
Exp/Cntr=0.5,0.3

Type RM Length L Ch R = 1 ,6586    ,59.3,58.7,58.7
XS GIS Cut Line= 4
2431964.83689881662905.5651595232431646.68738422  663074.6889223
2431411.89112031663131.2463947892431367.82090445663282.771301283
#Sta/Elev= 30
       0 1839.82    34.1 1832.05    70.3 1832.78   105.1 1826.14   153.4 1820.57
   237.9 1821.05   260.6 1819.89   274.6  1816.8   307.2 1818.83   357.5 1815.47
   367.1 1812.51   380.8  1802.7     389  1801.3   399.9 1794.05   405.5 1791.84
   409.6 1792.01   414.2 1794.62   417.9 1798.18     422 1799.78     450 1800.14
   473.2 1804.87   508.4 1806.78   526.2 1809.55   574.2 1819.63   617.2 1833.22
   672.3 1847.11   699.3 1855.95   730.6 1869.99   747.3 1881.56   759.6 1892.85
#Mann= 6 ,-1 , 0
       0     .05       0  339.62     .06       0   399.9    .045       0
   414.2     .06       0  441.34     .05       0     541      .1       0
Bank Sta=399.9,414.2
XS Rating Curve= 0 ,0
Exp/Cntr=0.5,0.3

Type RM Length L Ch R = 1 ,6527    ,373.1,362.8,354.5
XS GIS Cut Line= 4
2431916.22455095662837.0786358992431679.42682427663006.810931959
2431354.41178208663084.938182185 2431310.6971136663273.892681576
#Sta/Elev= 30
       0 1853.61    26.4 1853.61    85.5 1848.16   105.2 1841.53   128.5 1830.38
   149.5 1823.25   202.2 1815.82     216 1812.53   236.6 1815.12   267.6 1814.19
   301.9 1815.36   333.2 1813.28   341.4  1810.6   345.5 1808.07   353.8 1799.99
   368.3 1792.46   382.6 1790.05     3891792.439     399 1797.48   444.3  1796.9
     491 1801.43     544  1801.3     580 1806.84     617 1821.15     644  1824.9
   660.7 1832.65   685.1 1837.81   722.1 1850.86     767 1872.47   819.6    1904
#Mann= 6 ,-1 , 0
       0      .1       0   32.29     .05       0  300.96     .06       0
   368.3    .045       0     389     .06       0  500.16      .1       0
Bank Sta=368.3,389
XS Rating Curve= 0 ,0
Exp/Cntr=0.3,0.1

Type RM Length L Ch R = 1 ,6164    ,250.8,248,244.8
XS GIS Cut Line= 3
2431449.25057308662425.4425180852431365.42397684662788.810439934
2431226.51410131663114.132256136
#Sta/Elev= 30
       0 1987.48    42.5 1974.52   104.1 1960.39   141.1 1950.99   160.1 1945.22
   165.7 1943.11   173.9 1938.96   182.1 1937.71   186.2 1936.32   235.5 1914.52
   272.4 1896.03   301.2 1877.36   366.8    1826   379.5 1814.45   392.6 1803.99
   414.3 1785.19     423 1782.03   458.8  1778.6   475.2  1777.7   481.6 1779.27
   488.3 1784.28   492.6 1786.47   523.1 1786.62   544.8 1791.57   575.2 1800.72
   614.4 1809.25   631.8 1813.67   688.3 1832.28   710.1  1840.9   726.6 1848.52
#Mann= 5 ,-1 , 0
       0      .1       0  430.99     .06       0   458.8    .045       0
   481.6     .06       0  545.95      .1       0
Bank Sta=458.8,481.6
XS Rating Curve= 0 ,0
Exp/Cntr=0.3,0.1

Type RM Length L Ch R = 1 ,5916    ,125.3,115.2,110.2
XS GIS Cut Line= 3
     2431165.773       662386.242431114.21346309662912.966665713
2431176.08247758663033.207586086
#Sta/Elev= 30
       0 1904.18    44.9 1893.57    97.1 1883.17   117.2 1877.84   157.1 1870.17
   185.5 1867.53   237.8 1865.66   277.9 1862.24     286  1860.5   291.4 1857.68
   298.1 1853.04   334.2  1824.1   362.1 1800.49   390.5 1779.43   398.5 1774.81
   402.4 1773.84     417 1773.23   430.7 1771.27   434.7 1771.65   438.9 1773.87
   446.8 1779.36   450.8 1780.49   464.6 1782.05     487  1782.6     491 1783.49
     499 1787.13   531.1  1790.7   580.9 1798.97   648.4 1815.86   664.5 1821.11
#Mann= 5 ,-1 , 0
       0      .1       0  392.57     .06       0     417    .045       0
   438.9     .06       0  493.28      .1       0
Bank Sta=417,438.9
XS Rating Curve= 0 ,0
Exp/Cntr=0.5,0.3

Type RM Length L Ch R = 1 ,5801    ,87.9,91.4,93.2
XS GIS Cut Line= 3
2431059.81336032662381.5824129562430993.75427045662710.392113909
2431126.30022129663053.301187471
#Sta/Elev= 30
       0 1859.33    42.1 1846.77    91.1 1836.79   120.9 1832.43     136 1830.96
   212.7  1828.4   282.8 1828.84   303.2 1827.92   314.6 1826.27   319.6 1824.58
   331.6 1817.12   348.8 1801.94   361.6 1788.22   370.2  1780.5   382.9 1771.26
   387.4 1768.91   400.2 1767.46   408.8 1767.69   416.9 1769.27   430.3 1774.36
   438.8  1776.3   460.3 1778.76     486 1779.72   507.5  1783.4   526.7 1788.75
   548.9 1791.16   567.5  1794.8   630.4  1815.3   661.3 1823.14     703 1837.52
#Mann= 7 ,-1 , 0
       0      .1       0   11.63      .1       0  267.32      .1       0
   323.4     .06       0   387.4    .045       0   416.9     .06       0
  523.53      .1       0
#XS Ineff= 2 , 0
          380.45  1773.6  426.05          1774.3
Permanent Ineff=
       F       F
Bank Sta=387.4,416.9
XS Rating Curve= 0 ,0
Exp/Cntr=0.5,0.3

Type RM Length L Ch R = 1 ,5709    ,66.3,70.2,63.8
XS GIS Cut Line= 3
     2431042.257      662357.0342430909.15751575662722.709091006
2431098.15096405663077.711337094
#Sta/Elev= 30
       0 1856.63    45.4 1840.71   142.4 1822.43   159.5 1821.03   200.8  1815.1
   265.9 1808.62   299.9 1806.21     317  1806.5   325.5 1805.61   338.3 1799.44
   350.6 1791.81   361.1 1780.17   372.3 1772.47   407.5 1771.22     412 1768.56
   421.1 1759.85   424.5 1757.55   430.1 1755.79   435.1 1755.39   443.6 1756.47
   445.31757.492   455.5 1765.29   460.6 1770.19   470.9 1775.44   507.2 1779.85
   552.5 1782.28   605.3 1799.39   647.9 1811.01   733.7 1841.48   791.3 1857.71
#Mann= 7 ,-1 , 0
       0      .1       0   43.23      .1       0  164.99      .1       0
   368.5     .06       0   424.5    .045       0   445.3     .06       0
  584.67      .1       0
Bank Sta=424.5,445.3
XS Rating Curve= 0 ,0
Exp/Cntr=0.5,0.3

Type RM Length L Ch R = 1 ,5639    ,433.7,445.2,466.4
XS GIS Cut Line= 3
     2431007.393      662339.777 2430843.5982605 662712.63762084
2431019.19609848 663081.64025714
#Sta/Elev= 30
       0 1847.75    38.4 1836.01    60.2 1831.82      82 1824.82   103.9 1820.26
   112.6 1820.17   182.5 1809.47   303.4 1795.33   315.5 1791.28   329.8 1782.38
   349.7 1773.75   374.8  1769.9   392.2 1770.26   420.3 1768.97   431.9 1764.52
   445.2 1754.03   449.6 1751.87     454 1751.42     473  1753.6   480.6 1757.52
   495.3 1771.77   511.6 1783.16   524.9 1785.62   551.5 1785.62   609.4 1801.46
     638 1806.12   675.2 1824.46   768.6 1856.61   796.2 1870.43   815.9 1878.76
#Mann= 7 ,-1 , 0
       0      .1       0    71.5      .1       0  187.21      .1       0
  302.92     .06       0   445.2    .045       0     473     .06       0
  519.05      .1       0
Bank Sta=445.2,473
XS Rating Curve= 0 ,0
Exp/Cntr=0.3,0.1

Type RM Length L Ch R = 1 ,5194    ,301,300,296.5
XS GIS Cut Line= 3
2430872.80227774662193.226024962     2430569.693      662465.351
     2430277.963       662750.79
#Sta/Elev= 30
       0 1879.74   101.8 1830.59   146.2 1805.88   178.3 1790.02   196.3 1779.25
   209.4 1773.04   232.1 1766.47   277.4 1764.39   325.3  1758.9   339.7 1755.83
   376.5 1755.45   379.4 1754.47   384.4 1750.19   393.5 1738.01   396.4 1735.24
   400.6 1733.49   407.7 1733.08   417.1  1735.3   422.7 1739.18   424.7 1742.71
   428.3 1750.67   438.1 1776.29   439.4 1779.06     445 1786.65   481.2 1816.11
   532.1  1853.2   626.9 1913.18   758.4 2001.25   803.2 2029.88   815.5 2036.36
#Mann= 5 ,-1 , 0
       0      .1       0  234.87      .1       0  282.15    .055       0
   396.4    .045       0   417.1      .1       0
Bank Sta=396.4,417.1
XS Rating Curve= 0 ,0
Exp/Cntr=0.3,0.1

Type RM Length L Ch R = 1 ,4894    ,289.8,289.8,288.3
XS GIS Cut Line= 3
 2430647.9402195661892.821304874     2430394.765      662235.147
2430190.32672504662510.295222858
#Sta/Elev= 30
       0 1948.21    15.5  1943.8    57.3 1927.81      91 1911.55     112 1899.99
   211.5 1839.48     254 1811.63   325.5 1761.79   339.8    1753   355.8  1745.7
   365.5 1742.88   379.8 1741.32   390.6 1741.88   400.6 1741.17   405.6 1738.12
     417  1727.7   425.6 1725.69   435.4 1726.18   439.9 1727.77   459.3 1742.88
   471.4 1746.06   485.6 1754.81   519.7 1773.57   533.1 1779.32   579.6 1806.07
   651.5 1850.38   667.3 1861.15     674 1864.23   714.4 1888.66   768.6 1922.64
#Mann= 5 ,-1 , 0
       0      .1       0  366.33     .06       0     417    .045       0
   439.9     .06       0  504.94      .1       0
Bank Sta=417,439.9
XS Rating Curve= 0 ,0
Exp/Cntr=0.3,0.1

Type RM Length L Ch R = 1 ,4604    ,69.2,68.6,72.9
XS GIS Cut Line= 4
2430174.20125417661658.9328716062430160.67879189662069.114227575
2430088.91826406 662185.266231552430097.11161658662338.498535626
#Sta/Elev= 30
       0 1800.79      56 1795.79     128 1791.06   184.1 1785.69   228.1 1782.58
   248.8 1780.14   261.3 1777.53   284.1 1771.04   336.1  1749.7   375.3 1736.53
   388.2 1728.96   417.2 1728.86   421.9 1727.57   433.51719.561     436 1718.34
   445.4  1717.3   450.1 1717.42   456.7 1719.61   462.5 1721.28     475 1722.77
   482.9 1724.63   492.4 1730.21   517.7 1743.04   560.6 1769.46   572.6 1779.53
   593.3  1794.1   627.1 1819.36   636.7 1824.71   648.3 1832.44   700.4 1860.64
#Mann= 5 ,-1 , 0
       0      .1       0  158.92     .06       0   433.5    .045       0
   456.7     .06       0  499.21      .1       0
Bank Sta=433.5,456.7
XS Rating Curve= 0 ,0
Exp/Cntr(USF)=0,0
Exp/Cntr=0.5,0.3

Type RM Length L Ch R = 1 ,4536    ,69.9,63.8,64.1
XS GIS Cut Line= 4
2430086.18658656661663.8519329722430106.48871971662048.398219554
2430012.21549093662158.1628922272430042.92793504662336.038288104
#Sta/Elev= 30
       0 1741.41    31.1 1740.54    51.1 1738.47    79.1 1737.43   103.2 1735.83
   123.2 1735.92   171.8 1730.86   219.3 1728.03   385.1 1725.25   412.2 1722.95
     420 1720.64   425.41717.862   430.6 1715.98   439.9 1714.85   446.1 1716.05
   448.91718.006   454.7 1721.34   456.9 1722.04   467.5  1723.9   482.9 1732.26
   494.5 1736.93   511.5 1745.15     520 1750.29   529.8 1755.38   546.7 1768.07
     567 1780.54   591.3 1793.22   627.9 1810.54   668.5 1828.48   710.3 1843.59
#Mann= 4 ,-1 , 0
       0     .06       0   425.4    .045       0   448.9     .06       0
  534.61      .1       0
#XS Ineff= 2 , 0
          418.07  1722.5  454.21          1721.6
Permanent Ineff=
       F       F
Bank Sta=425.4,448.9
XS Rating Curve= 0 ,0
Exp/Cntr(USF)=0,0
Exp/Cntr=0.5,0.3

Type RM Length L Ch R = 1 ,4472    ,150.6,136.8,121.4
XS GIS Cut Line= 5
2429908.56033428661640.7603257132430040.39209867662021.151513807
2430003.67749272 662091.471858812429967.83679694662133.819039501
2429993.09963933 662337.70311133
#Sta/Elev= 30
       0 1792.71    57.3 1785.04     125 1769.65     142  1767.5   179.4 1757.24
   256.3 1738.12   305.2 1729.55   345.2 1728.16   362.1 1726.27   386.9 1725.33
     396 1723.14   402.6 1719.67   422.8 1713.32   436.1 1711.25   445.2 1711.06
   454.2  1711.2   458.21712.428   467.7 1718.71   472.2 1720.37   491.6  1721.8
   512.6 1721.78   523.1 1723.48   537.4  1729.8   542.5 1735.71   546.5 1739.27
   558.9 1746.94   570.7 1756.22     611 1775.95   675.5 1800.34   742.8 1822.36
#Mann= 8 ,-1 , 0
       0     .06       0  198.89      .1       0  290.25     .06       0
   422.8    .045       0   458.2     .06       0  550.16      .1       0
   622.4     .06       0  663.24      .1       0
Bank Sta=422.8,458.2
XS Rating Curve= 0 ,0
Exp/Cntr=0.5,0.3

Type RM Length L Ch R = 1 ,4335    ,260.5,253.8,243.8
XS GIS Cut Line= 3
2429795.53026963661781.0591760232429903.88013719662103.611790994
2429966.70165305662338.418571393
#Sta/Elev= 30
       0 1866.04      61 1837.96   110.6 1811.19   120.1 1805.23   148.3 1789.39
   183.4  1766.9   212.9 1745.72   246.7 1724.43   267.8 1708.54   273.3 1706.01
   284.6 1705.19   301.5 1706.25   305.7 1707.07   311.6 1709.19   318.4 1711.81
   331.1 1718.94   339.5 1720.88   348.5 1721.34   368.5 1720.98   387.7 1719.64
     391 1720.21   393.3 1721.12   397.4 1724.01   409.9 1735.33   414.3 1738.16
   463.7 1761.63   496.9 1773.93   518.4 1783.88   554.8 1797.84   583.3  1809.5
#Mann= 5 ,-1 , 0
       0      .1       0   273.3    .045       0   311.6     .06       0
  492.52      .1       0  543.78     .06       0
Bank Sta=273.3,311.6
XS Rating Curve= 0 ,0
Exp/Cntr=0.3,0.1

Type RM Length L Ch R = 1 ,4081    ,140.7,139.6,138.6
XS GIS Cut Line= 3
2429397.63874827661911.3141211812429762.18396438662277.488639402
2429825.75981016662418.932960194
#Sta/Elev= 30
       0 1983.85    24.2 1968.53    52.6 1953.28    67.1 1946.89    82.5 1942.85
    86.6 1938.47    96.6 1921.97   105.1 1910.25   112.3 1906.47   124.9 1892.82
   141.9 1880.34   163.1 1846.87   178.7 1835.27   191.3 1823.29     217 1810.78
     234 1789.15   245.4 1779.78   314.4 1740.96   347.4 1731.28   370.1 1727.93
   375.8 1725.45   396.5 1711.74   407.8 1701.49   428.4  1698.2   438.71698.917
   460.8 1707.61   548.9 1705.78   557.7  1707.2   623.5 1750.41   671.8 1777.66
#Mann= 5 ,-1 , 0
       0      .1       0  371.72     .06       0   407.8    .045       0
   438.7     .06       0  535.27      .1       0
Bank Sta=407.8,438.7
XS Rating Curve= 0 ,0
Exp/Cntr=0.3,0.1

Type RM Length L Ch R = 1 ,3942    ,397.3,397.7,395.6
XS GIS Cut Line= 3
2429295.28684686662042.6636724812429668.45841073662372.568968078
2429834.76312941662611.885514474
#Sta/Elev= 30
       0 1939.48    36.6 1910.31    95.4 1873.42   206.6 1792.55   325.7 1715.54
   335.6  1710.8   356.8 1705.06   394.4 1700.13   407.8 1693.07   421.1 1690.22
   436.2 1691.09   444.7 1695.06   453.2 1699.09   479.8 1699.22   495.8 1704.61
   501.4  1708.8   530.1 1776.97   539.9 1790.15   549.6 1797.08   570.4 1802.44
   588.6 1809.89     602  1816.1   649.3 1870.69   656.3 1873.44     671 1872.72
   676.7 1875.14   702.6 1912.98   726.4 1934.17   757.2 1944.19   789.5 1946.58
#Mann= 5 ,-1 , 0
       0      .1       0   407.8    .045       0   444.7      .1       0
   479.8     .06       0   588.6      .1       0
Bank Sta=407.8,444.7
XS Rating Curve= 0 ,0
Exp/Cntr(USF)=0,0
Exp/Cntr=0.3,0.1

Type RM Length L Ch R = 1 ,3544    ,441.2,450,459.8
XS GIS Cut Line= 3
     2428966.954      662229.009     2429270.767      662499.143
2429581.26624538662795.271631933
#Sta/Elev= 30
       0 1837.71      55 1831.39    74.7 1830.03    99.1 1824.96   168.3 1814.79
   187.1 1812.95   235.2 1798.87   255.7 1787.99   272.7 1775.04   294.1  1757.6
   331.6 1724.65     369 1698.47   386.5 1681.29   390.5 1679.82   406.2 1678.81
   417.7 1679.19   423.1 1680.68   452.5  1685.4   491.2 1684.77     528 1686.47
   533.7 1688.52   544.7 1694.81     562 1695.22   566.8 1696.64   576.1 1703.62
   603.2  1719.2   638.7 1735.91     661 1748.35   745.9 1800.71   835.6 1859.16
#Mann= 5 ,-1 , 0
       0      .1       0   386.5    .045       0   423.1      .1       0
  497.18     .06       0  620.16      .1       0
Bank Sta=386.5,423.1
XS Rating Curve= 0 ,0
Exp/Cntr=0.3,0.1

Type RM Length L Ch R = 1 ,3094    ,405.9,419.8,436.9
XS GIS Cut Line= 3
     2428877.411      662303.327     2428999.352      662831.149
2429097.45844255663205.123912881
#Sta/Elev= 30
       0 1818.48    32.4 1806.75      57 1800.52     135 1787.63   192.5 1773.14
   323.9 1722.93   336.2 1716.49   377.2 1690.46   401.9 1678.97   427.6 1671.33
   434.7 1670.44   463.5  1673.9   471.7 1669.47   475.8 1669.08   496.3 1674.45
   514.3 1674.83     521 1673.12   527.7 1668.52   533.2 1666.37     541  1666.2
   554.1 1667.52   560.7 1669.39   599.4 1698.97   607.6 1701.67   632.7 1702.26
   639.3 1705.95   653.1 1716.21   698.3 1734.59   876.4  1831.4   928.4 1857.57
#Mann= 5 ,-1 , 0
       0      .1       0  522.23     .06       0   527.7    .045       0
   560.7     .06       0  718.28      .1       0
#XS Ineff= 2 , 0
          504.04 1681.16
Permanent Ineff=
       F       F
Bank Sta=527.7,560.7
XS Rating Curve= 0 ,0
Exp/Cntr=0.3,0.1

Type RM Length L Ch R = 1 ,2674    ,336.8,330.2,321.1
XS GIS Cut Line= 3
     2428764.338      662283.379 2428693.0335998662660.234085829
     2428328.022      663023.163
#Sta/Elev= 30
       0 1816.76    72.8 1797.17   101.3 1787.28   146.1 1764.18   162.3 1757.26
   186.8 1748.86   223.4 1732.88   273.5 1706.37     313 1687.48   353.7 1665.69
   392.7 1660.62   460.1 1659.82     486 1656.97   499.6 1655.09   510.9 1655.88
   514.3 1657.56   522.8 1662.96   563.2 1673.84   579.4 1682.39   595.5 1682.45
   599.2 1683.48   636.9 1705.78   678.4 1723.53     722 1749.62   737.8 1752.85
   754.7 1763.21   802.8 1782.58   824.1 1790.19   842.4 1794.94   898.3 1804.86
#Mann= 5 ,-1 , 0
       0      .1       0     486    .045       0   514.3      .1       0
  551.85     .06       0  717.77      .1       0
#XS Ineff= 2 , 0
          459.87 1664.64
Permanent Ineff=
       F       F
Bank Sta=486,514.3
XS Rating Curve= 0 ,0
Exp/Cntr=0.3,0.1

Type RM Length L Ch R = 1 ,2344    ,446.8,450,451.6
XS GIS Cut Line= 3
     2428411.222      662189.768     2428356.522      662595.372
2428288.70935367663005.808629085
#Sta/Elev= 30
       0  1780.3   150.8 1735.11   186.8  1725.7   231.2 1706.83   267.5 1687.32
   291.7 1676.63   328.1 1654.72   372.5 1648.89   396.7 1648.98   408.8  1646.9
   412.8 1647.19     4181649.291   424.3 1653.07   429.1 1654.43   469.3 1655.58
   473.7  1656.5   489.9 1663.38   506.1 1664.28   510.1 1666.53   525.2 1678.45
   607.4 1729.44   633.1 1742.26   672.3 1759.77   684.5 1760.44   688.8 1762.07
   696.6 1767.21   716.9 1774.31   773.7 1789.71     798 1795.57   825.3 1800.43
#Mann= 5 ,-1 , 0
       0      .1       0   396.7    .045       0     418      .1       0
  429.94     .06       0   635.3      .1       0
Bank Sta=396.7,418
XS Rating Curve= 0 ,0
Exp/Cntr=0.3,0.1

Type RM Length L Ch R = 1 ,1894    ,422,414.5,407.9
XS GIS Cut Line= 3
     2428106.071      662046.449     2427945.167      662423.011
      2427786.26      662800.429
#Sta/Elev= 30
       0 1832.98    30.9  1816.6    61.4 1795.48   164.4 1723.03   183.2 1708.71
   210.1 1684.69   255.8 1653.29   274.5 1647.68   295.4 1643.74   353.3 1644.25
   374.7 1642.18   385.1 1639.18   400.7 1636.99   429.6 1639.31   444.1 1643.82
   457.1 1640.75   478.8 1644.44   500.5 1644.51   504.9 1647.89   515.1 1663.82
   522.2 1669.66     609 1714.52   634.2 1723.64   656.8 1728.65   692.2 1728.74
   717.5  1722.2   744.2 1713.09   760.9 1704.08   779.6 1699.91     819 1681.84
#Mann= 5 ,-1 , 0
       0      .1       0   385.1    .045       0   429.6      .1       0
  477.67     .06       0  592.27      .1       0
#XS Ineff= 2 , 0
                          444.47         1653.87
Permanent Ineff=
       F       F
Bank Sta=385.1,429.6
XS Rating Curve= 0 ,0
Exp/Cntr=0.3,0.1

Type RM Length L Ch R = 1 ,1479    ,395.7,394.8,391.5
XS GIS Cut Line= 3
2427583.89082351661793.1516108152427525.23078477662541.748066673
2427727.07334801662703.890251012
#Sta/Elev= 30
       0 1750.49    65.9 1762.72      94  1764.6   146.2 1762.13   177.6 1757.62
   202.4 1751.83   230.4 1748.44   278.6 1730.76   315.2 1721.74   342.8 1712.03
   386.9 1691.06   435.1 1665.94   459.1 1656.12   495.3 1638.52   507.3 1635.07
   523.6 1634.75   535.4 1630.72   547.4 1629.65   571.5 1627.61   585.11629.753
   595.6 1634.13   655.7  1630.7   675.8 1631.57   687.8 1633.79   699.9 1632.36
   763.1  1631.6   927.3 1634.84   942.7 1636.56   960.5 1641.24  1009.8 1659.21
#Mann= 6 ,-1 , 0
       0      .1       0   547.4    .045       0   585.1     .05       0
  655.98     .06       0  816.61     .05       0  964.99      .1       0
#XS Ineff= 2 , 0
                          608.62         1643.49
Permanent Ineff=
       F       F
Bank Sta=547.4,585.1
XS Rating Curve= 0 ,0
Exp/Cntr=0.3,0.1

Type RM Length L Ch R = 1 ,1085    ,126.4,127.8,126.1
XS GIS Cut Line= 4
 2427332.3335716661629.8934484392427161.15769124661885.714218442
2427193.26648985662334.5406875592427717.85323074662781.685801067
#Sta/Elev= 30
       0 1743.19    56.6 1708.54    82.6 1690.06   107.1  1675.2   148.9 1645.15
   174.9 1629.43   188.9 1622.77   204.3 1619.98     237 1619.23   465.4  1622.2
   540.6 1624.98   577.7 1622.99   589.7 1624.02   601.7 1620.43   625.8 1619.23
   638.41620.137   649.9 1626.16   653.9 1626.17   665.9 1622.12   685.9 1621.79
     706 1622.08   714.6 1623.76   817.5 1624.34   896.4 1627.22  1011.1  1629.3
  1176.2 1629.72  1285.3 1631.63  1363.4 1630.59  1400.9  1633.1  1447.1 1645.06
#Mann= 8 ,-1 , 0
       0      .1       0  161.55     .05       0   601.7    .045       0
   638.4     .06       0  820.44     .05       0 1102.03     .06       0
 1230.73     .05       0 1434.05      .1       0
#XS Ineff= 2 , 0
          543.74 1631.82  653.75         1633.54
Permanent Ineff=
       F       F
Bank Sta=601.7,638.4
XS Rating Curve= 0 ,0
Exp/Cntr=0.5,0.3

Type RM Length L Ch R = 1 ,957     ,53.5,54.1,54.8
XS GIS Cut Line= 4
 2427250.6989667661561.7407360782426954.94777062661892.052057896
2427226.35260964662507.9281925122427721.81399517662842.758029861
#Sta/Elev= 30
       0 1718.93    29.9 1696.33    71.6 1669.24   108.4 1642.07   142.4  1622.3
   162.2  1617.6   209.8 1616.65   293.8 1617.27   371.7 1615.65   577.6 1616.29
   669.4 1619.96   691.3 1622.12     700 1620.91   708.7 1617.04   721.9 1615.34
   739.3 1617.47   761.2 1624.64   787.4 1621.14   804.9 1620.39   891.4 1621.16
   952.1 1623.45  1052.2 1623.57  1200.3 1626.54  1271.4 1625.13    1332 1626.29
  1358.3 1625.69  1517.6 1630.16  1633.4 1627.74  1686.5 1630.18  1714.4 1637.45
#Mann= 5 ,-1 , 0
       0      .1       0  179.78     .05       0  598.29     .06       0
   708.7    .045       0   739.3     .06       0
#XS Ineff= 2 ,-1
    3.15   688.41620.863  769.01 1588.831620.746
Permanent Ineff=
       F       F
Bank Sta=708.7,739.3
XS Rating Curve= 0 ,0
Exp/Cntr=0.5,0.3
